--- GETOUTRN.prj (project) ---

Proj Title=GETOUTRN
Current Plan=p01
Default Exp/Contr=0,0
English Units
Geom File=g01
Flow File=f01
Plan File=p01
BEGIN DESCRIPTION:
---------- MODELED AS PART OF WVEMD CTP PROGRAM, 2023----------
Stream Name: Getout Run
Flood Zone:  AFH
Upshur County, WV
HEC-RAS Version: RAS 6.3
Vertical Datum: NAVD88
Projection: NAD 1983 StatePlane West Virginia S FIPS 4702 (US Feet)
Terrain: 1-meter LIDAR (FEMA Region III 3DEP collected 2016-2018)
Land Use: 2019 NLCD
Hydrologic Method:
WV SIR2010-5033 regression equations
Additional Model Notes:
Coincident peak with LIKANARV
END DESCRIPTION:
DSS File=dss
DSS Export Rating Curves= 0
DSS Export Rating Curve Sorted= 0
DSS Export Volume Flow Curves= 0
DXF OffsetX= 0
DXF OffsetY= 0
DXF ScaleX= 0
DXF ScaleY= 0

--- GETOUTRN.p01 (plan) ---

Plan Title=Floodplain
Program Version=6.30
Short Identifier=Floodplain
Geom File=g01
Flow File=f01
Subcritical Flow
K Sum by GR= 0
Std Step Tol= 0.01
Critical Tol= 0.01
Num of Std Step Trials= 20
Max Error Tol= 0.3
Flow Tol Ratio= 0.001
Split Flow NTrial= 30
Split Flow Tol= 0.02
Split Flow Ratio= 0.02
Log Output Level= 0
Friction Slope Method= 1
Unsteady Friction Slope Method= 2
Unsteady Bridges Friction Slope Method= 1
Parabolic Critical Depth
Global Vel Dist= 0 , 0 , 0
Global Log Level= 0
CheckData=False
Encroach Param=-1 ,0,0, 0
Computation Interval=0.1SEC
Output Interval=1SEC
Instantaneous Interval=Max Profile
Mapping Interval=1HOUR
Computation Time Step Use Courant=        0
Computation Time Step Use Time Series=    0
Computation Time Step Count To Double=0
Computation Time Step Max Doubling=0
Computation Time Step Max Halving=0
Computation Time Step Residence Courant=0
Run HTab= 0
Run UNet= 0
Run Sediment= 0
Run PostProcess= 0
Run WQNet= 0
Run RASMapper=-1
UNET Theta= 0
UNET Theta Warmup= 0
UNET ZTol= 0
UNET ZSATol= 0
UNET MxIter= 0
UNET Max Iter WO Improvement= 0
UNET MaxInSteps= 0
UNET DtIC= 0
UNET DtMin= 0
UNET MaxCRTS= 0
UNET WFStab= 0
UNET SFStab= 0
UNET WFX= 1
UNET SFX= 1
UNET Gravity=32.17405
UNET 1D Methodology=Finite Difference
UNET DSS MLevel= 1
UNET Pardiso=0
UNET DZMax Abort= 0
UNET Use Existing IB Tables= 0
UNET Froude Reduction=False
UNET Froude Limit= 0
UNET Froude Power= 0
UNET D1 Cores= 0
UNET WindReference=Eulerian
UNET WindDragFormulation=Hsu (1988)
UNET D2 Coriolis=0
UNET D2 Cores= 0
UNET D2 Theta= 1
UNET D2 Theta Warmup= 1
UNET D2 Z Tol= 0.01
UNET D2 Volume Tol= 0.01
UNET D2 Max Iterations= 20
UNET D2 Equation= 0
UNET D2 RampUpFraction=0.1
UNET D2 TimeSlices= 1
UNET D2 Turbulence Formulation=Non-Conservative (original)
UNET D2 Eddy Viscosity=0.3
UNET D2 Transverse Eddy Viscosity=0.1
UNET D2 Smagorinsky Mixing=0
UNET D2 BCVolumeCheck=0
UNET D2 Cores=0
UNET D2 SolverType=PARDISO (Direct)
UNET D2 Minimum Iterations= 3
UNET D2 Maximum Iterations= 30
UNET D2 Restart Number= 10
UNET D2 Relaxation Coeff=1.3
UNET D2 SOR Precondition Iterations= 10
UNET D2 ILUT Maximum Fill= 8
UNET D2 ILUT Tolerance=1E-08
UNET D2 Convergence Tolerance=0.00001
UNET D1D2 MaxIter= 0
UNET D1D2 ZTol=0.01
UNET D1D2 QTol=0.1
UNET D1D2 MinQTol=1
DSS File=dss
Write IC File= 0
Write IC File at Fixed DateTime=0
Write IC File at Sim End=0
Echo Input=False
Echo Parameters=False
Echo Output=False
Write Detailed= 0
HDF Write Warmup=0
HDF Write Time Slices=0
HDF Flush=0
HDF Compression= 1
HDF Chunk Size= 1
HDF Spatial Parts= 1
HDF Use Max Rows=0
HDF Fixed Rows= 1
Calibration Method= 0
Calibration Iterations= 20
Calibration Max Change=0.05
Calibration Tolerance=0.2
Calibration Maximum=1.5
Calibration Minimum=0.5
Calibration Optimization Method= 1
WQ AD Non Conservative
WQ ULTIMATE=-1
WQ Max Comp Step=1HOUR
WQ Output Interval=15MIN
WQ Output Selected Increments= 0
WQ Output face flow=0
WQ Output face velocity=0
WQ Output face area=0
WQ Output face dispersion=0
WQ Output cell volume=0
WQ Output cell surface area=0
WQ Output cell continuity=0
WQ Output cumulative cell continuity=0
WQ Output face conc=0
WQ Output face dconc_dx=0
WQ Output face courant=0
WQ Output face peclet=0
WQ Output face adv mass=0
WQ Output face disp mass=0
WQ Output cell mass=0
WQ Output cell source sink temp=0
WQ Output nsm pathways=0
WQ Output nsm derived pathways=0
WQ Create Restart=0
WQ Fixed Restart=0
WQ System Summary=0
WQ Write To DSS=0
Sorting and Armoring Iterations= 10
XS Update Threshold= 0.02
Bed Roughness Predictor= 0
Hydraulics Update Threshold= 0.02
Energy Slope Method= 1
Volume Change Method= 1
Sediment Retention Method= 0
Sediment TS Multiplier= 1
Warm Up Method= 0
XS Weighting Method= 0
Number of US Weighted Cross Sections= 1
Number of DS Weighted Cross Sections= 1
Upstream XS Weight=0
Main XS Weight=1
Downstream XS Weight=0
Number of DS XS's Weighted with US Boundary= 1
Upstream Boundary Weight= 1
Weight of XSs Associated with US Boundary= 0
Number of US XS's Weighted with DS Boundary= 1
Downstream Boundary Weight= 0.5
Weight of XSs Associated with DS Boundary= 0.5
Percentile Method= 0
Sediment Output Level= 3
Mass or Volume Output= 0
Output Increment Type= 1
Profile and TS Output Increment= 1
Transport Output Increment 1
XS Output Flag= 0
XS Output Increment= 10
Read HDF5 Sediment Hotstart= 0
Sediment Hotstart Type= 0
Write Gradation File= 0
Read Gradation Hotstart= 0
Write HDF5 File= 1
Write Binary Output= 1
Write DSS Sediment File= 0
DSS Sediment Output Type= 1
SV Curve= 0
Specific Gage Flag= 0
Subcell Erosion Methods= 0
Subcell Deposition Methods= 0
Advection Scheme= 1
Matrix Solver= 0
Implicit Weighting Factor= 1
Maximum Outer Loop Convergence Iterations= 5
Convergence Maximum Absolute= 0.001
Convergence RMSE= 0.0001
Grain Fractions Max Abs Error= 0.001
Max Subgrid Regions= 1
Max Subgrid Length Scale= 3.402823E+38
Initial Layer Thickness= 3.402823E+38
Min Layer Thickness= 3.402823E+38
Max Layer Thickness= 3.402823E+38
Number of Layers= 5

--- GETOUTRN.f01 (steady flow) ---

Flow Title=Flows
Program Version=6.31
Number of Profiles= 1
Profile Names=01pct
River Rch & RM=GETOUTRN,Main            ,10524
     679
River Rch & RM=GETOUTRN,Main            ,8472
     798
River Rch & RM=GETOUTRN,Main            ,5273
     926
River Rch & RM=GETOUTRN,Main            ,0
    1770
Boundary for River Rch & Prof#=GETOUTRN,Main            , 1
Up Type= 0
Dn Type= 1
Dn Known WS=1833.1
DSS Import GetInterval= 0
DSS Import GetPeak= 0
DSS Import FillOption= 0

--- GETOUTRN.g01 (geometry) ---

Geom Title=Geometry
Program Version=6.31

River Reach=GETOUTRN        ,Main
Reach XY= 30
2175234.45500004643649.6910000152175052.54100001643883.916000009
2174821.92200002      643897.5662174447.01800001644232.835999995
2174132.49600005644126.3540000172174124.56900002644294.703999996
     2173914.152644509.2989999952173917.32899998644836.069000021
2173353.01399998644925.5810000152173209.24500002645129.873999998
2173076.03600003645115.0789999962172827.90299998 645480.42400001
     2172384.492645635.6969999972172355.44599998645864.255999997
2172593.47800002646257.0729999992172169.41100003646563.068000019
      2171940.08      646873.7282171900.56000003647105.548999995
2171664.27500001647193.4590000062171792.16100003647402.244000003
2171560.74100003648116.995000005      2171590.53648334.680000022
2171340.99500002648314.019000009     2171072.889648495.132000014
2170770.47100003      648400.4412170442.09699999648434.008000001
2170004.72499998648752.5650000132169756.19100001648586.304000005
     2169618.146648600.6700000172169425.97297117 648783.99286519

Type RM Length L Ch R = 1 ,10524   ,63.7,63.7,63.7
XS GIS Cut Line= 5
2175113.40010439643596.8021049822175151.31219229643616.145006973
2175241.31365527643693.4133780012175265.98472209 643713.05885714
2175304.81880876643765.142220437
#Sta/Elev= 30
       0 2079.22     7.6 2077.11    16.6 2075.54    21.1 2074.47      39 2071.87
    54.2 2068.76    60.9 2067.95    70.1 2067.52    77.9 2067.74    85.9 2067.65
    91.1 2068.13    96.4 2068.31   101.7 2067.47     107 2067.05   111.7 2067.51
   123.3 2067.45     128 2067.12   131.8 2066.83   136.3 2067.08   143.9 2067.42
   154.5 2070.91   160.8 2072.06   168.7 2072.77   180.1 2072.58   192.7 2077.15
   202.9 2079.84   209.8 2080.74   232.8 2081.13     243 2082.79   257.7 2086.28
#Mann= 3 ,-1,0
       0      .1       0     128    .045       0   136.3      .1       0
Bank Sta=128,136.3
XS Rating Curve= 0 ,0
Exp/Cntr(USF)=0,0
Exp/Cntr=0.3,0.1

Type RM Length L Ch R = 1 ,10460   ,183.7,186,186.7
XS GIS Cut Line= 5
2175099.68345683643650.9243184692175140.80190154643687.017175491
2175198.82459573643733.6180794942175250.45108742643755.091045063
2175281.51835676643778.848368673
#Sta/Elev= 30
       0 2075.71     3.4 2074.95     9.5 2073.11    16.6 2071.79    27.3 2068.63
    32.6 2068.01    61.5 2066.15    64.6 2066.04    69.3  2066.3    72.9 2066.11
    77.3 2065.58    83.7 2064.45    89.9 2063.71    98.5 2064.46   102.9 2065.08
   115.5 2065.99   132.9 2069.17   143.6 2071.62   160.4 2074.91   172.7 2076.42
   181.8 2077.06   187.2 2077.93   193.5 2079.22   202.3 2079.39   207.4 2080.67
   210.6 2081.89   214.8 2083.19   217.4 2083.61     222 2083.93   224.2 2084.34
#Mann= 3 ,-1,0
       0      .1       0    83.7    .045       0    98.5      .1       0
Bank Sta=83.7,98.5
XS Rating Curve= 0 ,0
Exp/Cntr(USF)=0,0
Exp/Cntr=0.3,0.1

Type RM Length L Ch R = 1 ,10274   ,303.3,307,305.8
XS GIS Cut Line= 4
 2174964.4494609643690.2152767462174982.72432521643726.765005376
2175119.32893597643883.015095267 2175155.8786646643932.357228917
#Sta/Elev= 30
       0 2082.39     3.3 2081.97     7.8  2080.5    21.2  2072.1    30.1 2070.47
    34.6 2068.74    39.1 2066.05    49.1 2061.61    55.2 2057.52      60 2056.02
    63.4 2055.76    79.5  2056.2   107.8    2056   118.5 2057.41     140 2058.52
   158.5 2056.82   170.7 2057.27   182.8 2056.23   193.8 2056.22   219.4  2056.6
   224.7 2057.39   227.9 2059.99   235.3 2067.58   237.5 2068.87     246 2071.99
   256.1 2073.55     262  2076.8   276.7  2083.5   290.2 2088.45   309.8 2096.66
#Mann= 3 ,-1,0
       0      .1       0   182.8    .045       0   193.8      .1       0
Bank Sta=182.8,193.8
XS Rating Curve= 0 ,0
Exp/Cntr(USF)=0,0
Exp/Cntr=0.3,0.1

Type RM Length L Ch R = 1 ,9967    ,147.6,148.4,146.6
XS GIS Cut Line= 3
2174769.37090283643771.8550279622174869.66743167 643980.08972594
2174938.44219431644094.714330332
#Sta/Elev= 30
       0 2074.37     6.1 2072.35    14.8 2068.37    28.1 2065.73      37 2061.88
    54.7 2055.79    61.8 2055.16    76.9 2055.19    85.8 2055.78   103.6 2054.63
   125.9  2054.4   137.9 2053.71     148 2054.37   161.3 2055.99   174.6 2056.31
   185.9  2055.7   214.6  2057.8   223.5 2059.24   255.7 2066.13   265.1 2067.58
   274.6 2070.93   283.7 2071.21   288.4 2072.57   297.7 2077.18   306.6 2080.51
   316.4 2082.78   325.7 2086.19   330.4 2087.05   352.6 2094.63   364.8 2098.07
#Mann= 3 ,-1,0
       0      .1       0   125.9    .045       0     148      .1       0
Bank Sta=125.9,148
XS Rating Curve= 0 ,0
Exp/Cntr(USF)=0,0
Exp/Cntr=0.3,0.1

Type RM Length L Ch R = 1 ,9819    ,111.1,111.7,111.4
XS GIS Cut Line= 4
2174631.70452837643764.0087341532174636.00295103643843.959395716
2174800.20269682644122.497184389 2174841.4675544644180.955732628
#Sta/Elev= 30
       0 2081.38    17.2 2076.36    33.2 2072.96    57.3 2070.45      84  2063.5
    90.8 2063.18   100.1 2061.01   111.9 2060.88   127.7 2058.34   141.8 2054.78
   151.3 2053.26   174.9 2052.42   192.9 2053.32   211.5 2051.92   220.8 2053.34
   225.4 2053.36   239.4 2051.81   253.7 2051.43   259.3 2051.88   291.4 2053.85
   304.4 2057.12   313.6 2057.66   322.9 2059.64   336.9 2061.16   364.4 2070.35
   376.1 2072.69   406.7 2082.31   445.5 2093.16   459.8    2098     475  2101.4
#Mann= 3 ,-1,0
       0      .1       0   239.4    .045       0   259.3      .1       0
Bank Sta=239.4,259.3
XS Rating Curve= 0 ,0
Exp/Cntr(USF)=0,0
Exp/Cntr=0.3,0.1

Type RM Length L Ch R = 1 ,9707    ,82.9,82.9,82.6
XS GIS Cut Line= 4
2174600.93322577643897.9514847112174582.87983265643965.006944894
 2174678.3049106644130.0665391922174722.14886534644199.701055537
#Sta/Elev= 30
       0 2052.98    19.9 2049.38    28.2 2048.34    40.6 2047.49    48.9 2047.84
    53.1 2047.54    69.4  2045.1   111.2    2047   117.4 2046.19   125.1 2046.28
     136 2045.79     152 2045.94   159.9 2044.73     162 2044.51   164.9 2044.69
   167.9 2044.97   175.9 2044.56   185.2 2045.35   194.4 2045.51   215.9 2048.74
   231.4 2052.14   249.1 2057.61   254.5  2058.1   257.9 2058.94   263.7 2061.71
   266.6 2062.76   302.4 2074.08   320.5 2081.29   330.4 2085.93   342.4 2089.52
#Mann= 3 ,-1,0
       0      .1       0   159.9    .045       0   164.9      .1       0
Bank Sta=159.9,164.9
XS Rating Curve= 0 ,0
Exp/Cntr(USF)=0,0
Exp/Cntr=0.3,0.1

Type RM Length L Ch R = 1 ,9624    ,105.2,106.7,106.6
XS GIS Cut Line= 6
2174497.77097934643885.9158892932174474.76022499643951.780197507
2174512.38563092644011.4299557912174591.47668652644137.803707675
2174623.28504583644199.7010555372174662.83057364644244.404695659
#Sta/Elev= 30
       0 2053.46    11.9 2052.15    41.5 2050.03    54.3 2046.73    62.8 2045.21
    69.8 2044.97    80.9 2043.35    90.3  2043.3   109.3 2041.61     114 2042.72
   118.7 2042.96   128.2 2040.46   137.6 2039.28   170.7 2042.21   194.3 2041.08
   203.7 2041.16   228.5 2040.24   236.7 2039.11   245.5 2038.41   250.9  2039.1
   266.2 2039.47   279.2 2041.72   306.7 2048.16   320.2 2052.84     331 2054.96
   360.3 2067.52   372.4    2072     389 2079.75   408.6 2087.63   418.7 2092.57
#Mann= 3 ,-1,0
       0      .1       0   236.7    .045       0   250.9      .1       0
#XS Ineff= 2 , 0
          171.83 2060.87
Permanent Ineff=
       F       F
Bank Sta=236.7,250.9
XS Rating Curve= 0 ,0
Exp/Cntr(USF)=0,0
Exp/Cntr=0.3,0.1

Type RM Length L Ch R = 1 ,9518    ,115.7,116,115.7
XS GIS Cut Line= 3
2174373.79916849643964.3152303282174531.98112255644218.781852078
2174605.91399238644302.171251773
#Sta/Elev= 30
       0  2039.9    38.7 2039.76    66.2 2035.91    77.9 2035.17    81.1 2034.65
    90.5 2031.17    95.3 2030.69   137.6 2032.66   165.9 2034.97     180 2033.54
   189.4 2033.84   222.4  2031.1   234.7 2028.27   241.2 2026.03   250.6 2024.95
     255 2025.25   256.7 2025.99   260.1 2028.01   263.7 2031.82   269.1 2036.36
   274.2 2039.13   289.9 2045.54   302.8 2047.15     310 2051.67   318.9 2054.68
   348.2 2068.69   366.2 2078.97   377.7 2084.79   388.4 2089.34   411.1 2100.86
#Mann= 3 ,-1,0
       0      .1       0   241.2    .045       0   256.7      .1       0
Bank Sta=241.2,256.7
XS Rating Curve= 0 ,0
Exp/Cntr(USF)=0,0
Exp/Cntr=0.3,0.1

Type RM Length L Ch R = 1 ,9402    ,368.7,370,365.1
XS GIS Cut Line= 4
2174356.16633237644001.4168879122174329.42056478 644089.29583858
2174445.00048902644293.7099194822174490.85037633644351.022278613
#Sta/Elev= 30
       0  2038.7    12.3 2038.11    22.2 2036.27    49.9 2033.44    86.4 2031.55
   113.7 2027.52   123.9  2025.1   133.1  2026.1   142.3 2025.12   156.1 2025.43
   165.2 2026.72     179 2025.81   193.6 2026.42     225 2022.52   234.2 2022.88
     248 2021.69   261.7 2022.19     267 2021.29   272.9 2022.11   280.1 2023.25
   284.6 2025.42   298.5 2037.58   305.1 2041.99     311 2044.06   316.9 2044.72
   331.1 2051.91   346.5 2058.17   361.9 2068.62     383 2077.72   400.1 2087.72
#Mann= 3 ,-1,0
       0      .1       0   261.7    .045       0   272.9      .1       0
Bank Sta=261.7,272.9
XS Rating Curve= 0 ,0
Exp/Cntr(USF)=0,0
Exp/Cntr=0.3,0.1

Type RM Length L Ch R = 1 ,9032    ,277.5,281.5,279.4
XS GIS Cut Line= 4
2173957.70151106643977.2263197042174051.04920789644011.799540755
2174280.38490753644343.7024628392174380.64724858644400.172057221
#Sta/Elev= 30
       0 2052.81      24 2042.47    42.4 2038.21    53.8 2034.03    70.9 2028.82
    82.8 2027.12    92.2 2023.94     133 2019.46   149.8 2019.53   187.6 2017.83
     200  2018.9   227.9 2018.52   233.6 2017.56   237.4 2017.02   243.82017.545
   251.9    2019   266.5 2018.31     286 2018.61   302.6 2019.82   377.4 2019.57
   412.4 2020.49   441.6 2020.24   456.1    2021   472.3 2020.85   486.6 2024.52
   518.6 2035.08   530.3 2036.56     544  2040.9   585.4  2047.8     618 2057.52
#Mann= 3 ,-1,0
       0      .1       0   233.6    .045       0   243.8      .1       0
Bank Sta=233.6,243.8
XS Rating Curve= 0 ,0
Exp/Cntr(USF)=0,0
Exp/Cntr=0.3,0.1

Type RM Length L Ch R = 1 ,8750    ,285,277.8,261.5
XS GIS Cut Line= 5
2173908.30731239644189.349870031 2174027.1772725644295.483762986
2174137.55652117 644454.684602422174199.11417908644473.788703152
2174294.63468274644467.420669574
#Sta/Elev= 30
       0 2043.51    45.1 2037.33    67.8 2033.02    74.9 2032.14    84.8  2029.5
    98.9 2027.54   110.3 2027.25   175.1 2021.27   182.2  2021.2   204.4 2017.32
   210.2 2017.27   215.9 2015.88   218.8 2014.91   221.7 2014.71   227.4  2015.8
   233.2 2017.37   238.3  2017.6   296.4  2016.4   307.9 2017.63     322 2020.31
   333.8 2021.27   352.6 2020.48   406.1 2023.53   418.6 2023.39   434.1 2025.14
   454.7 2025.78     468 2029.68   478.7  2030.3   486.8 2031.56   513.3 2038.63
#Mann= 3 ,-1,0
       0      .1       0   215.9    .045       0   227.4      .1       0
Bank Sta=215.9,227.4
XS Rating Curve= 0 ,0
Exp/Cntr(USF)=0,0
Exp/Cntr=0.3,0.1

Type RM Length L Ch R = 1 ,8472    ,169.1,169.7,170.5
XS GIS Cut Line= 5
2173759.09841976644461.0409989162173872.66168522644535.334723985
2173988.34762854644533.2120461262174133.61020088644528.679818857
2174301.44261276644659.511378743
#Sta/Elev= 30
       0 2052.28    61.6 2036.25      76 2031.38   120.8 2021.06   131.8 2019.01
   143.2 2017.89   163.2 2013.99   171.2 2012.58   175.2 2012.62   183.2 2014.02
   231.2 2015.16   243.2 2017.46   247.2 2017.62   266.8 2016.93   303.3 2017.19
   327.3 2018.71   367.3 2018.33   391.3 2019.89   410.6 2019.07   435.5 2019.94
   455.9  2018.1   475.6 2019.86   481.1 2021.17   501.7 2023.93   516.6 2023.95
   536.9 2026.17   561.4  2026.9   577.5 2028.17   592.7 2030.28   609.5 2031.01
#Mann= 3 ,-1,0
       0      .1       0   163.2    .045       0   183.2      .1       0
Bank Sta=163.2,183.2
XS Rating Curve= 0 ,0
Exp/Cntr(USF)=0,0
Exp/Cntr=0.3,0.1

Type RM Length L Ch R = 1 ,8302    ,349.1,366.2,375.7
XS GIS Cut Line= 5
2173723.99852915 644647.388238462173807.85740754 644699.80003745
2173920.54277537 644699.80003745 2173980.8163442644743.039771617
2174062.05463264644858.345729396
#Sta/Elev= 30
       0  2020.6    10.1 2019.94    18.8 2021.22    23.8 2021.23    36.3 2019.17
    48.7 2018.56    56.8 2019.34    66.2 2018.35    89.8 2018.65   123.2 2017.56
   135.2 2016.39   155.2 2012.16   163.2 2010.65   171.2 2012.17   187.2 2013.76
   203.2  2017.8   226.6 2020.31   245.6 2023.73   255.1    2023   275.1 2024.18
     285 2025.78   312.4 2027.67   317.7 2027.09   322.6 2027.47   356.9 2032.88
   381.9 2038.54     393 2041.56   400.9 2044.56   410.3 2045.79   426.8 2051.82
#Mann= 3 ,-1,0
       0      .1       0   155.2    .045       0   171.2      .1       0
Bank Sta=155.2,171.2
XS Rating Curve= 0 ,0
Exp/Cntr(USF)=0,0
Exp/Cntr=0.3,0.1

Type RM Length L Ch R = 1 ,7936    ,329.3,327.1,322.8
XS GIS Cut Line= 4
2173646.69112564644670.9735480052173688.62056483644762.694196239
2173723.99852915644942.2046077812173772.47944322645056.200270585
#Sta/Elev= 30
       0 2024.28     6.8 2022.72    15.6 2022.23    48.1 2017.43    59.6 2016.76
    77.2 2017.41    90.4 2015.47   119.6 2014.84   127.8 2014.02     140 2011.22
   156.4 2010.14   184.9 2010.22   201.2 2013.03   205.3 2012.45   213.5 2009.46
   217.5 2008.51   221.6 2008.42   229.8 2009.37   237.9 2010.48   241.7 2012.05
   254.2 2020.33   262.4  2023.8   279.7 2026.28   289.3 2026.66   317.5 2031.32
   321.8 2033.15   347.9 2040.61   369.6 2049.46   386.9 2054.79   407.7 2063.21
#Mann= 3 ,-1,0
       0      .1       0   213.5    .045       0   229.8      .1       0
Bank Sta=213.5,229.8
XS Rating Curve= 0 ,0
Exp/Cntr(USF)=0,0
Exp/Cntr=0.3,0.1

Type RM Length L Ch R = 1 ,7609    ,256,260.4,256.9
XS GIS Cut Line= 2
2173328.72481716644791.9234277432173501.81634829645123.822237437
#Sta/Elev= 30
       0 2032.83     9.4 2028.11    19.5 2026.96    30.2  2022.8      42 2020.34
    64.6 2013.48    78.1 2012.04    87.1 2012.63   100.7 2009.29   118.7 2006.38
   127.7 2008.31   132.2 2008.54   143.1 2006.41   150.3 2005.66   160.6 2006.31
   186.4 2008.72   206.4 2007.53     218 2008.26     227 2007.22   240.5  2009.8
     245 2009.64   258.6 2011.15   272.1 2011.14   285.6 2013.02   294.6 2015.53
   312.7 2019.09   344.5 2022.51   362.3    2026   371.3 2029.06   374.3 2029.11
#Mann= 3 ,-1,0
       0      .1       0   143.1    .045       0   160.6      .1       0
Bank Sta=143.1,160.6
XS Rating Curve= 0 ,0
Exp/Cntr(USF)=0,0
Exp/Cntr=0.3,0.1

Type RM Length L Ch R = 1 ,7349    ,87.3,87.5,85.1
XS GIS Cut Line= 4
2173187.07167016644972.6033788562173244.72464905645060.393142165
2173277.48202342645152.1137903982173348.02999239645216.862624052
#Sta/Elev= 30
       0 2016.03    21.4 2012.78      39 2010.77    48.5    2010    58.1 2008.83
    64.8  2008.7    77.3  2007.6    86.8 2005.18     104 2003.95   110.1 2003.05
   118.6  2002.4   133.32000.111   139.6 1999.71   144.62000.082   148.3 2000.43
   156.8  2002.5   161.1 2002.57   169.6 2000.72   174.1 2000.03   178.1 2000.62
   186.6 2002.57     204 2004.03   216.4 2006.62   250.4 2005.97   260.4 2006.99
   265.8 2007.84   278.7 2011.07     290 2013.45   292.9 2013.84   298.2 2013.79
#Mann= 3 ,-1,0
       0      .1       0   133.3    .045       0   144.6      .1       0
Bank Sta=133.3,144.6
XS Rating Curve= 0 ,0
Exp/Cntr(USF)=0,0
Exp/Cntr=0.3,0.1

Type RM Length L Ch R = 1 ,7261    ,254,248.4,239.8
XS GIS Cut Line= 2
2173148.07103467644985.1809625022173216.13129691645245.658509351
#Sta/Elev= 30
       0 2017.89     4.1 2016.72    29.6 2011.42    41.3 2009.51    53.7 2006.97
    70.3    2004    82.7 2002.87    99.2 2000.94   111.6 1997.47   119.9  1994.4
   132.3 1991.41   137.8 1990.88   144.7 1989.76     153 1990.99   157.4 1991.12
   161.2 1992.03   165.4 1993.81   173.6 1995.33   180.4 1994.05   190.2  1993.5
   194.3 1993.96   198.4  1995.1   202.6 1995.79     215 1997.07   219.7 1997.29
   243.9  1997.1   253.6 1997.55   260.5  1997.6   264.6 1997.99   269.2 1998.95
#Mann= 3 ,-1,0
       0      .1       0   137.8    .045       0     153      .1       0
Bank Sta=137.8,153
XS Rating Curve= 0 ,0
Exp/Cntr(USF)=0,0
Exp/Cntr=0.3,0.1

Type RM Length L Ch R = 1 ,7013    ,85.7,86.4,86.4
XS GIS Cut Line= 3
2172952.50162848645176.5845861442173108.20004945645258.732219291
2173213.27260348645244.404143742
#Sta/Elev= 30
       0 2023.02     9.1 2019.96    17.7 2016.53    23.9 2015.76    26.8 2014.96
    31.3 2012.75    40.3 2009.69    44.9 2007.24    53.9 1999.76      72 1987.09
    76.5  1984.9      81 1983.22    85.6 1982.43    90.1 1982.19   103.7 1981.05
   108.2  1981.2   112.7 1982.19   118.6 1983.15   130.5 1983.78   139.8 1985.41
   151.2 1988.24   155.6 1988.99   171.5  1989.7   184.1 1991.61   208.3 1993.12
   220.4 1994.68   236.6 1995.47   246.7 1996.97   272.9 1997.25   282.1 1998.32
#Mann= 3 ,-1,0
       0      .1       0    90.1    .045       0   112.7      .1       0
Bank Sta=90.1,112.7
XS Rating Curve= 0 ,0
Exp/Cntr(USF)=0,0
Exp/Cntr=0.3,0.1

Type RM Length L Ch R = 1 ,6926    ,99.4,101.3,103.2
XS GIS Cut Line= 4
2172919.93948807645256.4169280712172953.37166435 645270.74500362
2173047.93696297645325.1916907062173148.23349181645358.623866987
#Sta/Elev= 30
       0 2012.96     4.6 2011.72       9 2010.02      19  2005.1      22 2004.11
    26.4 2003.53    28.2 2002.91    30.7 2001.79    40.2 1995.51    51.9 1989.72
    57.3  1987.5    73.3 1982.04    81.1 1980.04    87.1 1978.92    92.9 1978.44
    98.11978.957   108.8 1980.43   113.5 1981.44   127.3 1985.95   131.9 1987.17
   145.7  1989.5   154.2 1990.12   162.6 1991.29     171 1991.47   183.7 1992.36
   186.8 1994.01   187.9 1994.28     196 1993.27   204.8 1993.44   251.2 1997.76
#Mann= 3 ,-1,0
       0      .1       0    87.1    .045       0    98.1      .1       0
Bank Sta=87.1,98.1
XS Rating Curve= 0 ,0
Exp/Cntr(USF)=0,0
Exp/Cntr=0.3,0.1

Type RM Length L Ch R = 1 ,6825    ,119.3,121.5,122.3
XS GIS Cut Line= 3
2172856.98112482645309.3580862312172909.51740184645352.342312878
 2173026.0524163645450.728431648
#Sta/Elev= 30
       0 2013.74     4.1 2012.88    10.7 2012.07    14.5 2010.86    18.7  2009.2
    33.4 2002.96    36.3 2001.38    43.9 1996.56    50.6 1993.49    56.6  1992.4
      61 1990.64    67.5 1986.36    70.4 1984.81    73.2 1983.68    81.8 1981.02
    90.2 1979.61    97.5 1978.96   104.4 1977.41     108 1976.86   112.6 1976.69
   117.4 1977.41     130 1981.29   135.6 1983.83   139.4 1985.16   155.5  1988.5
   181.1 1988.72   198.1 1989.57   205.6 1989.46   212.3  1989.7   220.4 1989.05
#Mann= 3 ,-1,0
       0      .1       0   104.4    .045       0   117.4      .1       0
Bank Sta=104.4,117.4
XS Rating Curve= 0 ,0
Exp/Cntr(USF)=0,0
Exp/Cntr=0.3,0.1

Type RM Length L Ch R = 1 ,6704    ,118,121.2,124.4
XS GIS Cut Line= 2
2172778.39214139645375.809636562 2172936.5621795645551.953542634
#Sta/Elev= 30
       0 2009.42     7.2 2007.27    12.6 2006.61      18 2005.33    23.3 2003.06
    34.1 1999.38    44.6 1993.84    50.6 1989.36    53.2 1988.38    56.6    1988
      61 1986.04    67.4 1980.32    70.2 1979.01    74.5 1978.33    84.4 1978.19
   104.4 1975.37   110.4 1974.18   114.7 1973.85   125.5 1975.34   130.9 1976.93
   138.2 1981.02   143.9 1983.31   155.2  1985.2   160.9 1985.63   168.5 1985.05
   182.3 1985.05   194.8 1986.13   211.5 1986.31   216.9 1987.26   236.7 1989.18
#Mann= 3 ,-1,0
       0      .1       0   104.4    .045       0   125.5      .1       0
Bank Sta=104.4,125.5
XS Rating Curve= 0 ,0
Exp/Cntr(USF)=0,0
Exp/Cntr=0.3,0.1

Type RM Length L Ch R = 1 ,6582    ,125.8,127.3,128.7
XS GIS Cut Line= 3
2172702.90189593645391.9861177322172776.59475459645587.901278567
2172782.26072179645600.304588009
#Sta/Elev= 30
       0 2013.62    14.1 2008.81    31.2 2002.14    39.7 2000.38      44 1998.89
    52.6 1993.97    65.4 1984.99    69.7 1982.24    73.9  1979.2    78.2 1975.69
    82.5 1973.55    86.7 1973.19    99.6 1973.81   108.1 1973.21   112.4 1973.68
   125.2 1974.39   129.5 1973.72   136.9 1971.74   142.3 1970.84   146.6 1971.33
   147.9  1971.8   159.4 1976.92   163.4 1978.25   167.9 1979.31   172.2 1979.83
   180.8  1980.6   193.6 1980.98   202.1 1980.84     210 1981.24     223 1979.91
#Mann= 3 ,-1,0
       0      .1       0   136.9    .045       0   147.9      .1       0
Bank Sta=136.9,147.9
XS Rating Curve= 0 ,0
Exp/Cntr(USF)=0,0
Exp/Cntr=0.3,0.1

Type RM Length L Ch R = 1 ,6455    ,75.6,74.5,73.6
XS GIS Cut Line= 4
2172612.81690035 645445.561372082172624.42264154645501.268929815
 2172633.7072345645574.7719573812172641.44439529 645621.19492216
#Sta/Elev= 30
       0 2005.41     7.8 2003.35      16 2001.88      20 2000.38    28.2 1996.88
    39.7 1994.01    44.6  1992.1    49.9 1988.66    56.8 1983.11    60.8 1979.45
    64.9 1974.97    68.9 1971.56    72.9 1969.53      77 1968.81      81 1968.62
      85 1968.89    89.1  1969.4    97.1 1970.79   105.2 1971.36   109.2  1972.7
   113.3 1973.63   117.3 1973.96   129.4 1974.11   141.5 1972.81   145.6 1972.78
   153.7 1974.13   161.8 1974.78   169.9 1975.28     174 1975.31   178.1 1974.98
#Mann= 3 ,-1,0
       0      .1       0    72.9    .045       0    89.1      .1       0
#XS Ineff= 2 , 0
                          126.42         1977.33
Permanent Ineff=
       F       F
Bank Sta=72.9,89.1
XS Rating Curve= 0 ,0
Exp/Cntr(USF)=0,0
Exp/Cntr=0.3,0.1

Type RM Length L Ch R = 1 ,6381    ,194,187.8,177
XS GIS Cut Line= 3
2172532.75163296645446.8413476832172578.20722784  645636.1009476
2172695.61421554645666.729579562
#Sta/Elev= 30
       0 2005.07    18.9 1999.12    27.1 1995.89    47.7 1993.74    51.8 1992.68
    55.9 1990.64    67.8 1986.76    72.3 1984.79    76.5 1982.22    88.8 1972.99
    92.9 1970.51      97 1968.89    99.91968.437   109.4 1968.22   111.61968.381
   125.8 1970.01     134 1971.34   146.4 1971.87   157.4 1971.78     167 1972.88
   187.2 1972.77   200.8 1973.45   225.6 1972.47   242.1 1972.29   271.1 1973.17
   279.4 1972.43   287.6 1973.22     300 1973.57   308.3  1974.3     316 1973.69
#Mann= 3 ,-1,0
       0      .1       0    99.9    .045       0   111.6      .1       0
#XS Ineff= 2 , 0
                           202.7          1978.9
Permanent Ineff=
       F       F
Bank Sta=99.9,111.6
XS Rating Curve= 0 ,0
Exp/Cntr(USF)=0,0
Exp/Cntr=0.3,0.1

Type RM Length L Ch R = 1 ,6193    ,186.3,180.9,171.2
XS GIS Cut Line= 5
2172274.20556375645593.4249043872172355.92866133645606.160971542
2172432.34506425 645657.105240162172610.65000442 645658.16657909
2172786.83226673645731.398965229
#Sta/Elev= 30
       0 2011.93    30.3 2002.21    38.4 1996.97    42.5 1995.99    54.6 1995.17
    62.7 1991.41    92.6 1982.17    99.5 1978.59     111  1969.7     116 1967.21
   121.5 1965.79   128.3  1965.5   139.9 1967.19   160.3    1970   218.2 1967.99
   234.4 1968.71   246.4 1970.35   266.4 1969.74   298.4 1971.73   310.4 1970.72
   353.3 1971.98   397.8 1971.28   423.8 1972.06   449.8 1975.82   462.8 1976.78
   493.1 1977.76     517 1977.34   524.6 1978.33   536.4 1982.03   543.7  1983.1
#Mann= 3 ,-1,0
       0      .1       0     116    .045       0   139.9      .1       0
Bank Sta=116,139.9
XS Rating Curve= 0 ,0
Exp/Cntr(USF)=0,0
Exp/Cntr=0.3,0.1

Type RM Length L Ch R = 1 ,6012    ,102.5,101.1,99.4
XS GIS Cut Line= 5
2172213.70924477645791.8952842142172298.61635913 645801.44733458
2172407.93426887645788.7112674252172623.38607157645804.631351369
2172722.09059202645852.391603199
#Sta/Elev= 30
       0 2019.15    34.7 2007.25    50.8 2003.38    62.9 1998.71    70.9 1993.65
      79 1993.31      83 1992.25      87 1989.71    99.1 1978.57   107.1 1972.46
   123.3 1964.46   130.4 1963.69   139.81963.722   148.4 1965.89   167.6 1967.18
   183.7 1966.71   191.7 1967.25     276 1964.18   334.4 1964.42   351.2  1963.3
   364.2 1963.31   380.2 1968.35   400.3 1971.41   412.4 1972.01   421.3 1976.09
   434.6  1977.8   448.5 1982.78   484.4 1991.83   511.4 1997.06   521.2 1998.06
#Mann= 3 ,-1,0
       0      .1       0   130.4    .045       0   139.8      .1       0
Bank Sta=130.4,139.8
XS Rating Curve= 0 ,0
Exp/Cntr(USF)=0,0
Exp/Cntr=0.3,0.1

Type RM Length L Ch R = 1 ,5911    ,97.7,98.6,98.6
XS GIS Cut Line= 6
2172287.13556312645911.7649457552172338.20082438 645900.15920456
2172417.89358058645880.8163025692172607.45402009645877.721438251
 2172641.4975276645873.0791417732172689.46792454645891.648327684
#Sta/Elev= 30
       0 1996.96     5.2 1995.76    13.4  1995.5    17.5 1994.28    29.8 1987.28
    46.2 1976.41    54.4 1969.76    58.5 1967.17    66.7 1963.69    70.9 1962.66
      83 1962.07    89.6 1962.66   107.9 1965.04   144.7 1965.68   177.7 1962.05
   188.7 1962.61   208.7 1961.63   216.7 1962.71   224.7 1962.44   248.7 1963.66
   288.7 1961.56   292.7 1961.81   300.7 1963.75   312.7 1970.38   340.8  1978.4
   344.9 1979.96   348.9  1982.7   352.9  1984.5   378.3 1992.24   409.8 1999.66
#Mann= 3 ,-1,0
       0      .1       0    70.9    .045       0    89.6      .1       0
Bank Sta=70.9,89.6
XS Rating Curve= 0 ,0
Exp/Cntr(USF)=0,0
Exp/Cntr=0.3,0.1

Type RM Length L Ch R = 1 ,5812    ,307.6,307.4,307.8
XS GIS Cut Line= 2
2172274.42005253646004.6428009492172680.05921548645936.582538708
#Sta/Elev= 30
       0 2004.49    26.1 1995.99    34.2 1992.45    46.4 1991.32    74.8 1983.01
    84.4 1978.16   103.2 1966.55   115.3 1961.24   127.5 1959.47   131.6 1959.49
   139.3 1961.21   147.8 1963.61   155.9 1964.17   176.2 1962.97   212.7 1962.97
   220.8 1961.39   228.9 1961.92   237.2 1960.79   249.2 1961.86   281.6 1960.49
   289.7  1962.3   301.9 1961.04   318.1 1961.94   334.4  1966.8   348.4 1972.84
   354.6 1976.16   362.8 1982.61     379 1984.79   391.1 1992.07   411.3 2001.07
#Mann= 3 ,-1,0
       0      .1       0   115.3    .045       0   139.3      .1       0
Bank Sta=115.3,139.3
XS Rating Curve= 0 ,0
Exp/Cntr(USF)=0,0
Exp/Cntr=0.3,0.1

Type RM Length L Ch R = 1 ,5505    ,222.6,231.2,237.5
XS GIS Cut Line= 5
2172365.35240018646166.885415966 2172428.7197471646182.204994343
2172545.00927388646199.6136061352172633.44502178 646197.52457272
2172708.65022472646192.650161418
#Sta/Elev= 30
       0 1979.53    19.4 1974.25    27.6 1973.04    49.6 1968.33    64.6 1963.02
    76.8 1956.78    80.8 1956.23      97 1955.98   109.1 1957.39   129.4 1957.88
   145.5 1956.45   153.6    1957   165.8 1959.19   182.8 1959.44   193.9 1960.71
     210 1957.45     218 1956.76   221.31955.811     226 1955.22   228.6 1955.81
   239.1 1959.06     242  1960.8   246.9 1965.25     262 1975.27     274  1980.4
   285.4  1987.2     293 1989.81     310 1997.17   338.1 2005.21   346.6 2009.59
#Mann= 3 ,-1,0
       0      .1       0   221.3    .045       0   228.6      .1       0
Bank Sta=221.3,228.6
XS Rating Curve= 0 ,0
Exp/Cntr(USF)=0,0
Exp/Cntr=0.3,0.1

Type RM Length L Ch R = 1 ,5273    ,85.5,86.3,86.9
XS GIS Cut Line= 4
 2172354.4493016646232.2822937512172420.15795381646289.388965725
2172517.57322114 646400.618342732172535.49886423646485.055336971
#Sta/Elev= 30
       0 1979.71    12.9 1976.09    18.2  1975.3    23.5    1974    39.4 1969.38
    55.3 1966.01    69.9 1961.42    76.5 1958.47    81.8 1956.79    89.8 1955.95
   118.7 1956.71     124 1955.73   135.7 1954.53   146.4 1951.64   152.1 1951.29
   156.91951.533   172.1 1955.92   177.2 1956.34   187.8 1955.25   198.4 1956.66
   208.5 1956.52     223 1958.14   243.7 1959.76   276.4 1963.77   288.2 1966.02
   292.7 1967.34   300.9 1971.54   304.9 1972.52   309.1 1972.46   321.2 1970.36
#Mann= 3 ,-1,0
       0      .1       0   146.4    .045       0   156.9      .1       0
Bank Sta=146.4,156.9
XS Rating Curve= 0 ,0
Exp/Cntr(USF)=0,0
Exp/Cntr=0.3,0.1

Type RM Length L Ch R = 1 ,5187    ,132.1,132.3,132.8
XS GIS Cut Line= 4
2172329.79116204646328.6342409662172368.37143115646356.046537438
2172427.76474017646433.7147107762172490.71149504646504.275992436
#Sta/Elev= 30
       0 1976.08     7.8 1973.63    12.7 1971.75    16.4 1970.59    35.5 1965.89
      48 1961.84    50.8 1960.54    60.2 1955.11    65.1 1952.87    68.9 1952.08
    73.9 1952.23      79 1951.84      84 1950.85      89 1950.59    93.7 1950.85
    99.7 1951.57   109.2 1952.73   129.3 1953.22   133.6 1954.06   139.3 1956.56
   144.4 1957.91   157.7 1959.47   176.5 1960.93   187.3 1961.95   199.8 1962.66
   205.8 1963.68   211.8 1964.15   224.8 1965.68   232.7 1966.95   239.7 1968.35
#Mann= 3 ,-1,0
       0      .1       0      79    .045       0    99.7      .1       0
Bank Sta=79,99.7
XS Rating Curve= 0 ,0
Exp/Cntr(USF)=0,0
Exp/Cntr=0.3,0.1

Type RM Length L Ch R = 1 ,5055    ,99.2,98.2,97.1
XS GIS Cut Line= 4
2172252.81181879646426.3240414792172280.38705987 646457.03283268
 2172339.9245122646539.1318458912172370.00659337646585.508387705
#Sta/Elev= 30
       0 1979.53     9.2 1975.95      20 1972.19      23 1970.92    29.9 1967.11
    36.1 1964.02    46.4 1957.81    47.7  1956.9    52.7 1952.73    55.5 1950.78
    56.3 1950.44    58.4 1949.79    61.3 1949.31    64.1 1949.25    68.2 1949.37
      76 1950.41    84.2  1951.7    88.6 1952.08    90.9 1952.09   100.7 1951.15
   104.2 1951.36   107.1  1951.9   112.8 1953.57   115.6 1954.17   125.5 1955.89
   143.1  1956.6   154.7 1958.18   164.2 1960.02   190.6 1962.14     198 1962.49
#Mann= 3 ,-1,0
       0      .1       0    56.3    .045       0      76      .1       0
Bank Sta=56.3,76
XS Rating Curve= 0 ,0
Exp/Cntr(USF)=0,0
Exp/Cntr=0.3,0.1

Type RM Length L Ch R = 1 ,4957    ,117.5,114,109.4
XS GIS Cut Line= 3
2172171.99235579646484.2979080692172248.59024768646572.037311501
2172282.01478232 646617.29970216
#Sta/Elev= 30
       0 1979.67     3.6 1977.64     6.5 1976.42     9.3 1975.68    12.1 1974.53
    14.9 1973.11    22.4 1968.75    29.1 1964.18    31.9  1962.4    37.6 1959.19
    43.6 1954.95    48.9  1951.6    51.8  1950.3    54.3 1949.43    59.6 1948.93
      66 1948.66    70.2 1948.69    75.5 1949.37    80.8 1950.93    85.4 1952.08
    96.7 1955.64   102.1  1956.3   108.5 1956.81   115.8 1957.95   122.7 1958.33
   132.8 1959.24   142.8 1959.87   151.3 1959.89   157.7 1960.16   172.7 1959.83
#Mann= 3 ,-1,0
       0      .1       0    54.3    .045       0    75.5      .1       0
Bank Sta=54.3,75.5
XS Rating Curve= 0 ,0
Exp/Cntr(USF)=0,0
Exp/Cntr=0.3,0.1

Type RM Length L Ch R = 1 ,4843    ,97.2,96.7,95.4
XS GIS Cut Line= 4
2172091.53044727646581.5745561892172117.22555827646601.629276973
2172185.53695094646636.0983283222172261.36886391646648.632528812
#Sta/Elev= 30
       0 1967.81     5.9 1964.94    20.1 1959.32    26.2 1957.91    31.5 1954.97
    35.9 1952.85    40.4 1951.32    53.8 1947.23    58.3  1946.5    62.8 1946.61
    66.81947.294    71.7 1948.86    82.1 1949.59    89.7 1951.64    98.6 1954.49
   102.9 1955.42   107.6 1956.21   111.8 1956.52   115.8 1956.47     128 1957.05
   133.2  1957.1   136.7 1957.34   144.2 1958.21   152.3 1958.21   156.4 1958.51
   160.4 1959.42   164.5 1959.94   172.6 1960.14   180.7 1960.76     186 1960.89
#Mann= 3 ,-1,0
       0      .1       0    53.8    .045       0    66.8      .1       0
Bank Sta=53.8,66.8
XS Rating Curve= 0 ,0
Exp/Cntr(USF)=0,0
Exp/Cntr=0.3,0.1

Type RM Length L Ch R = 1 ,4746    ,106.2,109.7,111.5
XS GIS Cut Line= 5
2172044.45108498646662.8967275072172069.57902341646683.912821469
2172135.82540655646711.3251179412172212.12296507646704.928915431
2172256.89638264646699.446456137
#Sta/Elev= 30
       0 1961.99      16 1955.49    20.5 1954.46    30.9 1952.74    36.1 1951.68
    39.9 1950.26    44.2 1947.73    46.5 1946.77    48.6 1946.15    57.1 1945.91
    61.5 1946.18    65.9 1946.88    70.2  1947.8    78.9 1947.84    83.2  1948.3
    90.8 1950.53    98.8 1953.48   104.8 1954.79   108.8 1955.08   117.9 1954.91
   132.7 1955.37   144.9 1955.23     153 1956.07     161 1956.22   172.6 1957.56
   193.2 1957.78   197.2 1958.04   205.2 1959.23   209.3 1959.59   226.1 1960.13
#Mann= 3 ,-1,0
       0      .1       0    46.5    .045       0    65.9      .1       0
Bank Sta=46.5,65.9
XS Rating Curve= 0 ,0
Exp/Cntr(USF)=0,0
Exp/Cntr=0.3,0.1

Type RM Length L Ch R = 1 ,4636    ,110.8,109.7,109.5
XS GIS Cut Line= 4
2171978.14872271646743.4784687862172068.19811662646810.090349213
2172129.05341478646808.8567958722172203.88898415646832.294309355
#Sta/Elev= 30
       0 1970.62     8.4 1966.14      17 1961.09    22.4  1958.2    37.3 1951.11
    42.3 1948.91    48.4 1945.66    49.9 1945.08    52.3 1944.52    62.7 1944.22
    68.4 1944.61    72.2 1945.77    76.8 1948.42    82.1 1949.93    87.1 1949.94
    92.1 1950.82   102.8 1951.73     112 1953.45     116 1953.45     124 1952.63
     128 1952.49     156 1952.62   176.1 1953.31     198 1952.59   213.9 1952.94
   227.5 1952.51   230.6 1952.69   233.1 1953.11   242.7 1955.18   251.3 1957.96
#Mann= 3 ,-1,0
       0      .1       0    48.4    .045       0    72.2      .1       0
Bank Sta=48.4,72.2
XS Rating Curve= 0 ,0
Exp/Cntr(USF)=0,0
Exp/Cntr=0.3,0.1

Type RM Length L Ch R = 1 ,4527    ,157.3,154.1,152.8
XS GIS Cut Line= 4
2171917.58197393646813.3649229952171916.10170992646836.309015142
2171993.81557041646885.5277934582172127.30540635646965.846639286
#Sta/Elev= 30
       0 1969.62     7.8 1968.38    27.8 1963.91    32.5 1961.26    38.2 1956.34
    46.9 1948.01    51.5 1945.06    52.7 1944.55    54.5 1943.97    56.2 1943.73
    64.3 1943.38      73 1943.91    76.9 1944.44    89.4  1946.5    94.1  1948.1
    98.8 1948.77   117.7 1948.61   136.4 1949.62   139.8 1949.29   145.6 1948.31
   150.4 1948.01   159.7 1949.73   171.8 1951.11   186.4 1951.54   197.1 1952.23
   211.1 1953.47   225.1 1954.12   241.8 1955.95   261.7 1959.03   270.8 1961.06
#Mann= 3 ,-1,0
       0      .1       0    52.7    .045       0    76.9      .1       0
Bank Sta=52.7,76.9
XS Rating Curve= 0 ,0
Exp/Cntr(USF)=0,0
Exp/Cntr=0.3,0.1

Type RM Length L Ch R = 1 ,4373    ,89.1,92.2,92.8
XS GIS Cut Line= 5
2171851.87417187646968.1520633382171898.13242216646994.796815509
2171945.87093647647014.0402476322171990.64892276 647027.73268972
2172035.05684304647058.448167917
#Sta/Elev= 30
       0 1957.13     2.1 1956.81       5    1956     9.6 1954.12    14.2 1953.14
    18.8 1952.89    32.7 1952.83    41.9 1951.54    51.1 1950.61    55.6 1949.67
    59.9 1948.47      66 1945.31    68.5 1944.29    72.8 1943.35    77.1 1943.63
    85.8 1945.35    98.7 1948.07   107.3 1949.23   111.4 1949.35   119.8 1948.66
     124 1948.68   128.4 1949.21   136.5  1950.9   144.9 1951.67   153.5 1953.35
   159.6 1952.95   162.4 1952.99   188.3 1954.16   196.9 1955.58   205.7 1956.45
#Mann= 3 ,-1,0
       0      .1       0      66    .045       0    85.8      .1       0
Bank Sta=66,85.8
XS Rating Curve= 0 ,0
Exp/Cntr(USF)=0,0
Exp/Cntr=0.3,0.1

Type RM Length L Ch R = 1 ,4280    ,100,106.6,109.8
XS GIS Cut Line= 5
2171819.44542514646984.5344639262171850.53096934647029.682516215
2171857.19215738647065.2088524432171925.28430182647102.955584685
2171996.70704028647143.662844946
#Sta/Elev= 30
       0 1957.41     5.6 1956.24    15.4 1953.72    20.2 1952.78    35.5 1951.89
    49.3 1951.78    70.6 1951.14    76.4 1950.41    93.1 1947.13    99.1 1946.68
   104.9 1946.03   112.7 1945.55   117.2  1945.1     131  1943.5   137.3 1942.36
   140.2 1941.78   144.7 1941.49   149.3 1941.47     152 1941.81   154.9 1942.44
   158.4  1943.6   167.5 1947.39   172.1 1948.63   181.3 1950.06   190.2 1950.95
   204.4 1950.89   210.7 1951.77   225.4 1952.81   242.9 1952.95     251  1953.8
#Mann= 3 ,-1,0
       0      .1       0   137.3    .045       0   154.9      .1       0
Bank Sta=137.3,154.9
XS Rating Curve= 0 ,0
Exp/Cntr(USF)=0,0
Exp/Cntr=0.3,0.1

Type RM Length L Ch R = 1 ,4174    ,146.9,146,145
XS GIS Cut Line= 4
2171738.77102192647028.6545632672171800.94212502647115.167762764
2171847.57044132647172.1579271292171883.83690955647188.810897236
#Sta/Elev= 30
       0    1958     2.4 1956.99     7.1  1955.6    24.3 1952.87    30.2  1952.3
    49.9 1951.32    59.8 1950.57    64.7  1949.4    70.2 1946.03      73 1944.61
    75.9 1943.57    79.5 1942.74    84.5 1942.27    99.2 1943.67   113.1 1943.45
     118 1942.96   124.3 1941.65   130.6 1939.58   136.9 1938.91   147.2 1939.53
   160.8 1939.75     166 1940.82   171.2 1942.49   176.3 1944.54   185.2 1946.79
   189.6 1947.55   199.5 1948.56   205.5  1949.6   211.6 1950.07   220.1 1951.82
#Mann= 3 ,-1,0
       0      .1       0   130.6    .045       0   147.2      .1       0
#XS Ineff= 2 , 0
          105.63  1947.5
Permanent Ineff=
       F       F
Bank Sta=130.6,147.2
XS Rating Curve= 0 ,0
Exp/Cntr(USF)=0,0
Exp/Cntr=0.3,0.1

Type RM Length L Ch R = 1 ,4028    ,87.4,79.3,70.4
XS GIS Cut Line= 3
 2171652.8422827647131.7244968662171705.83938921 647195.22965036
2171766.14644145647221.271332008
#Sta/Elev= 30
       0  1960.3     3.4    1960     5.2 1959.69     7.1 1958.94     9.1 1957.57
    12.3 1954.56    17.5 1949.35    23.9 1944.15    27.9 1941.06    30.2 1939.64
    31.8 1938.86    34.6  1937.8    36.4 1937.34    42.7 1936.31    48.8 1936.19
      54  1936.5    57.4  1937.3    60.2 1938.36    64.4 1940.37    65.9 1940.89
    69.6 1941.83    74.4 1942.52    80.1 1942.69    89.6 1942.66   101.2 1943.21
   119.4 1943.41   128.8 1943.18   137.5 1943.27   146.3 1942.64   148.4  1942.6
#Mann= 3 ,-1,0
       0      .1       0    36.4    .045       0    57.4      .1       0
Bank Sta=36.4,57.4
XS Rating Curve= 0 ,0
Exp/Cntr(USF)=0,0
Exp/Cntr=0.3,0.1

Type RM Length L Ch R = 1 ,3948    ,126.2,119.3,108.9
XS GIS Cut Line= 3
2171610.35322317647239.5461963232171679.34083596647239.089324715
2171773.45638718 647235.89122346
#Sta/Elev= 30
       0 1955.25     1.8 1955.11     5.8 1953.85     9.8 1951.08    13.8 1947.26
    17.8 1943.72    21.8 1940.89    25.8 1939.15    29.8 1938.18    37.8 1936.63
    43.7 1935.75    49.8 1934.79    53.8 1934.64    57.8 1934.91    61.8 1935.92
    65.8 1937.19    73.8 1940.72    77.8 1941.56    81.8 1941.93    93.8 1942.23
   101.8 1942.64   105.8 1942.61   109.8 1942.79   125.8 1942.35   133.9 1942.71
   137.9 1942.39   141.9  1941.8   145.9  1941.4   152.9 1941.49   163.2 1941.96
#Mann= 3 ,-1,0
       0      .1       0    43.7    .045       0    61.8      .1       0
Bank Sta=43.7,61.8
XS Rating Curve= 0 ,0
Exp/Cntr(USF)=0,0
Exp/Cntr=0.3,0.1

Type RM Length L Ch R = 1 ,3829    ,110.9,121.2,128.7
XS GIS Cut Line= 4
2171676.82522192 647374.620005172171722.46669554647305.129833613
2171773.86475143647273.879815635 2171840.8878163647266.889680034
#Sta/Elev= 30
       0 1940.96     1.7 1941.31     6.1 1941.21    11.3 1939.11    16.1 1936.58
      28 1934.34    35.2 1932.37    38.1 1931.47      41 1931.12    49.6 1932.48
    57.1 1935.12    63.9 1936.63      79 1937.04    85.1 1937.85    89.8 1939.08
   103.9 1939.76   108.5 1940.34   122.6 1939.72     132 1939.96     146 1942.05
   153.7 1943.65   157.7 1943.62   165.7 1941.65   167.9 1941.81   173.8 1942.74
   185.8  1945.6   197.9 1945.45   201.9 1946.32   205.9 1947.85   210.7 1948.49
#Mann= 3 ,-1,0
       0      .1       0    35.2    .045       0    49.6      .1       0
Bank Sta=35.2,49.6
XS Rating Curve= 0 ,0
Exp/Cntr(USF)=0,0
Exp/Cntr=0.3,0.1

Type RM Length L Ch R = 1 ,3708    ,81.3,87.8,93.5
XS GIS Cut Line= 3
2171697.66991678647402.5295975742171851.63564863647405.270827221
2171904.17588354647430.398765654
#Sta/Elev= 30
       0 1937.69    22.5 1935.99    38.5 1934.28    58.5 1934.62    74.5 1933.46
    78.5 1932.28    87.6 1928.62    90.5 1927.59    94.5 1926.97    99.4 1928.46
   105.8 1931.43   110.5 1932.94   113.9  1934.7     118 1937.37   130.5 1947.15
   134.3 1949.46   142.5 1953.78   150.5 1956.39   154.3 1958.18     159 1961.36
   163.3 1963.65   167.9 1965.21   181.2 1968.78   190.1 1971.97   194.5 1972.79
   199.3 1974.57   203.4 1977.92   205.3 1980.65   207.8 1984.78   212.2 1996.59
#Mann= 3 ,-1,0
       0      .1       0    87.6    .045       0    99.4      .1       0
Bank Sta=87.6,99.4
XS Rating Curve= 0 ,0
Exp/Cntr(USF)=0,0
Exp/Cntr=0.3,0.1

Type RM Length L Ch R = 1 ,3620    ,50.3,47.5,44.1
XS GIS Cut Line= 3
2171681.60631105647418.7256960732171771.53234963647495.329358564
2171802.24782782647506.431338636
#Sta/Elev= 30
       0 1939.87     3.8 1939.96    12.1 1936.73    14.9 1935.89    17.7 1935.45
    43.3 1934.89    50.7 1935.57    51.8 1935.41    55.9 1934.29    66.4 1929.55
    71.6  1927.6    74.5 1926.92    77.3 1926.36      83 1925.88    85.8 1926.25
    88.7 1927.13    92.7 1928.78      98 1931.38   102.5 1931.98   108.5 1931.97
   113.7  1932.4   117.1 1932.92   123.1 1934.48   127.3 1936.17   131.6  1938.9
   135.8 1942.36   140.1 1944.24   144.3 1944.75   148.6 1944.36   150.8 1943.69
#Mann= 3 ,-1,0
       0      .1       0    74.5    .045       0    88.7      .1       0
Bank Sta=74.5,88.7
XS Rating Curve= 0 ,0
Exp/Cntr(USF)=0,0
Exp/Cntr=0.3,0.1

Type RM Length L Ch R = 1 ,3573    ,92,89,87
XS GIS Cut Line= 4
2171665.64677052647462.3893668692171684.56125508647498.162413765
 2171751.9955044647524.0670339312171778.72249347647538.458489578
#Sta/Elev= 30
       0 1935.14     5.4 1934.95    21.3 1932.93    30.6 1932.51    39.4 1931.69
    44.3 1931.73    45.6 1931.55    48.6 1930.92    51.8 1929.64    57.2 1927.17
      60 1926.33    61.5 1925.99    65.8 1925.67    70.4 1925.09    74.3 1924.53
    78.6 1924.44    85.8 1925.08    87.2 1925.27    91.5 1926.59    95.8 1928.57
     100 1929.46   104.3 1929.63     122 1929.06   125.5  1930.8   126.5 1931.56
   128.4  1933.2   131.1 1935.85   135.6 1939.65   140.2 1941.77   143.1  1941.6
#Mann= 3 ,-1,0
       0      .1       0    70.4    .045       0    85.8      .1       0
Bank Sta=70.4,85.8
XS Rating Curve= 0 ,0
Exp/Cntr(USF)=0,0
Exp/Cntr=0.3,0.1

Type RM Length L Ch R = 1 ,3484    ,54.4,55.4,58.9
XS GIS Cut Line= 5
2171601.03610054647572.7671219612171660.61672692647591.640488082
 2171735.7401254647593.4908180942171778.29771568647602.742468153
2171813.82405191647607.553326184
#Sta/Elev= 30
       0 1935.56     3.3 1934.84    11.7 1931.88    15.9 1931.16    21.9 1930.86
    28.5 1931.02    37.9 1930.47    45.3  1929.2    50.6 1928.59      57 1928.17
      62 1928.15    66.1 1927.78    74.1  1924.5    78.1 1923.48    86.1 1923.24
    93.3 1924.42    98.1 1925.22   102.1  1925.6   106.5 1925.65     122 1926.66
   126.1 1926.34   130.1 1926.81   134.3 1928.16     155 1931.63   162.7 1932.04
     179 1931.81   195.2 1933.88   199.2  1935.4   207.3 1939.61     217 1944.01
#Mann= 3 ,-1,0
       0      .1       0    74.1    .045       0    93.3      .1       0
Bank Sta=74.1,93.3
XS Rating Curve= 0 ,0
Exp/Cntr(USF)=0,0
Exp/Cntr=0.3,0.1

Type RM Length L Ch R = 1 ,3428    ,53.9,54.3,56.3
XS GIS Cut Line= 4
2171601.03610054 647627.166824312171659.50652892647640.859266398
2171745.36184147647641.5993984032171800.87174182 647642.70959641
#Sta/Elev= 30
       0 1930.94     3.2 1930.49     8.8 1930.44    15.5  1930.1    34.2 1927.99
    44.2 1927.16    48.4 1927.12    56.6 1928.01    60.7 1928.15    68.7 1927.55
    72.7 1927.05    80.7 1925.41    84.6 1924.98    92.7    1923   100.8 1921.84
   104.7 1921.44   108.7 1921.34   112.9 1921.47   116.7 1921.83   120.9 1922.65
   124.5 1923.73   140.7  1927.8   145.1 1928.32   153.3 1928.42   164.7 1928.98
   168.7  1929.5   176.7 1931.74   184.7 1933.64   196.7 1938.03   201.4 1940.06
#Mann= 3 ,-1,0
       0      .1       0   100.8    .045       0   116.7      .1       0
Bank Sta=100.8,116.7
XS Rating Curve= 0 ,0
Exp/Cntr(USF)=0,0
Exp/Cntr=0.3,0.1
